--- Clear Fork A.prj (project) ---

Proj Title=Clear Fork A
Current Plan=p01
Default Exp/Contr=0,0
English Units
Geom File=g01
Flow File=f01
Plan File=p01
BEGIN DESCRIPTION:
END DESCRIPTION:
DSS Export Rating Curves= 0
DSS Export Rating Curve Sorted= 0
DSS Export Volume Flow Curves= 0
DXF OffsetX= 0
DXF OffsetY= 0
DXF ScaleX= 0
DXF ScaleY= 0

--- Clear Fork A.p01 (plan) ---

Plan Title=Floodplain
Program Version=4.00
Geom File=g01
Flow File=f01
K Sum by GR=0
Std Step Tol=0.01
Critical Tol=0.01
Num of Std Step Trials=20
Max Error Tol=0.3
Flow Tol Ratio=0.001
Split Flow NTrial=30
Split Flow Tol=0.02
Split Flow Ratio=0.02
Log Output Level=0
Friction Slope Method=1
Unsteady Friction Slope Method=2
Unsteady Bridges Friction Slope Method=1
Global Log Level=0
CheckData=False
Run HTab=0
Run UNet=0
Run PostProcess=0
UNET Theta=0
UNET Theta Warmup=0
UNET ZTol=0
UNET ZSATol=0
UNET MxIter=0
UNET MaxInSteps=0
UNET DtIC=0
UNET DtMin=0
UNET MaxCRTS=0
UNET WFStab=0
UNET SFStab=0
UNET WFX=0
UNET SFX=0
UNET DSS MLevel=0
UNET DZMax Abort=0
UNET Convert EG Bridges=0
UNET Use Existing IB Tables=0
UNET Froude Limit=0
UNET Froude Power=0
Write IC File=0
Echo Input=False
Echo Output=False
Write Detailed=0

--- Clear Fork A.f01 (steady flow) ---

Flow Title=NFF Regression Equation
Program Version=4.00
Number of Profiles=1
Profile Names=P100yr
River Rch & RM=Clear Fork A,Main      ,38218.5
2769.935
River Rch & RM=Clear Fork A,Main      ,36503.2
3060.253
River Rch & RM=Clear Fork A,Main      ,32329.2
3116.571
River Rch & RM=Clear Fork A,Main      ,32024.5
3693.907
River Rch & RM=Clear Fork A,Main      ,27136.4
4077.418
River Rch & RM=Clear Fork A,Main      ,17541.1
4440.060
Boundary for River Rch & Prof#=Clear Fork A,Main      ,1
Up Type=0
Dn Type=3
Dn Slope=0.010251

--- Clear Fork A.g01 (geometry) ---

Geom Title=Geometry
Program Version=4.00

River Reach=Clear Fork A    ,Main
Reach XY= 30
     1770602.229      144286.787     1769944.436      144546.117
     1769135.469      145511.029     1768422.886      145111.419
     1768066.293       144523.65     1767452.559      144604.597
     1767043.259      144233.203     1765979.742      144299.204
      1765611.49      145630.499     1764882.774      146089.166
     1764826.271      146591.873     1763398.852      148852.021
     1762092.567      149604.419     1761267.984      151438.215
     1760364.274      152210.047     1759363.756      152469.439
     1759394.246      155349.503     1758866.277      156396.163
     1758159.832      156643.918     1757082.599      155719.385
     1755633.731      155075.173     1755232.609      155298.917
      1755075.28      156041.444     1753126.264      157453.231
     1752323.316      159129.882     1752322.504       160081.07
     1754088.109       161532.31     1754403.889      163282.966
     1754828.182      163977.712     1754493.608      164983.854

Type RM Length L Ch R = 1 ,38218.5 ,119.6,119.7,119.9
XS GIS Cut Line= 2
     1770188.495      143925.949     1770603.654      144835.715
#Sta/Elev= 30
       0 1628.08    10.1 1628.08    30.3 1618.46    60.6 1600.73   141.4 1548.64
   161.6 1536.37   181.8 1525.06   232.3 1498.41   272.7  1479.2   323.2 1457.67
   363.6 1441.14   373.7 1437.58   383.8 1435.47   393.9 1434.62   444.5  1433.6
   464.7 1432.37   474.8 1428.42     495 1411.01   505.1 1406.24   510.2 1406.16
   515.2  1397.8   520.2 1406.76   545.5 1410.73   555.6 1411.56   666.7 1414.57
   737.4 1419.49   747.5 1421.27   757.6 1425.28   828.3 1468.13    1000 1569.57
#Mann= 3 , 0 , 0
       0      .1       0   510.2    .045       0   520.2     .06       0
Bank Sta=510.2,520.2
XS Rating Curve= 0 ,0
Exp/Cntr=0.3,0.1

Type RM Length L Ch R = 1 ,38098.7 ,211.9,211.2,210.5
XS GIS Cut Line= 2
     1770244.033      144332.572      1770376.65      144628.271
#Sta/Elev= 21
     9.8 1426.95    19.6  1424.2    29.5 1423.31    68.7 1420.78    78.6 1419.95
    88.4 1418.46    98.2 1414.69     108 1408.89   117.8 1405.04   122.7 1404.72
   127.7 1397.75   132.7 1405.25   137.5 1406.08   147.3 1408.76   157.1 1410.82
   166.9 1411.68   216.1 1413.41   265.2 1414.97   304.4 1416.32   314.3 1416.88
   324.1 1418.91
#Mann= 3 , 0 , 0
     9.8      .1       0   122.7    .045       0   132.7     .06       0
Bank Sta=122.7,132.7
XS Rating Curve= 0 ,0
Exp/Cntr=0.3,0.1

Type RM Length L Ch R = 1 ,37887.5 ,322.5,314.7,306.8
XS GIS Cut Line= 2
     1770052.163      144404.258     1770189.619      144682.936
#Sta/Elev= 24
      10 1435.08    30.1 1426.67    50.1    1418    60.1 1413.35    70.2 1408.09
    80.2 1403.38    85.2 1402.29    90.2  1397.7    95.2  1401.4   100.2  1401.6
   110.3  1403.1   120.3 1404.71   130.3 1405.91   140.3 1406.62   150.4 1407.03
   170.4 1407.63   230.5 1409.03   240.6 1409.66   250.6 1410.71   260.6 1411.96
   280.7  1414.5   290.7 1415.93   300.7 1418.26   310.7 1422.47
#Mann= 3 , 0 , 0
      10      .1       0    85.2    .045       0    95.2     .06       0
Bank Sta=85.2,95.2
XS Rating Curve= 0 ,0
Exp/Cntr=0.3,0.1

Type RM Length L Ch R = 1 ,37572.9 ,469.6,467.7,465.7
XS GIS Cut Line= 3
     1769734.606      144547.182     1769792.315      144617.033
     1770010.738      144809.094
#Sta/Elev= 26
    10.1 1453.43    30.2 1445.26    60.4 1432.74    70.5 1428.68    80.5 1424.72
   110.7 1413.17   120.7 1408.82   130.7 1403.83   140.8  1400.2   145.8 1399.66
   150.8 1397.68   155.8 1399.61   160.8 1400.11   170.8 1401.89   180.9  1403.3
   190.9 1404.03     211 1404.97     231 1405.65   281.2 1406.86   291.2 1407.46
   301.2  1408.6   331.3 1413.54   341.3 1415.52   351.4 1418.93   361.4  1424.3
   381.5 1435.96
#Mann= 3 , 0 , 0
    10.1      .1       0   145.8    .045       0   155.8     .06       0
Bank Sta=145.8,155.8
XS Rating Curve= 0 ,0
Exp/Cntr=0.3,0.1

Type RM Length L Ch R = 1 ,37105.2 ,315.2,315.5,315.3
XS GIS Cut Line= 2
     1769449.617      144950.316     1769688.753      145121.665
#Sta/Elev= 23
     9.8 1431.45    19.6 1426.23    29.4 1421.42    39.2 1416.89      49 1412.93
    58.8 1409.46    68.6  1406.4    78.5 1403.16    88.3 1399.44    98.1  1396.6
   102.9 1396.16   107.9 1395.71   112.9 1395.91   117.7  1396.1   127.5 1397.34
   137.3 1398.73   147.1 1400.01   156.9 1401.08   166.7 1401.77   264.8 1405.54
   274.6 1406.14   284.4 1408.42   294.2 1412.55
#Mann= 3 , 0 , 0
       0     .08       0   102.9    .045       0   112.9     .08       0
Bank Sta=102.9,112.9
XS Rating Curve= 0 ,0
Exp/Cntr=0.3,0.1

Type RM Length L Ch R = 1 ,36789.7 ,271.5,286.6,301.7
XS GIS Cut Line= 3
     1769261.955       145187.41     1769504.223      145338.205
     1769728.295      145355.151
#Sta/Elev= 30
     9.8 1425.12    19.7 1419.47    29.5 1414.62    39.4 1410.69    49.2 1407.41
      59 1404.65    68.9 1402.94   137.8 1397.51   167.3  1394.6   172.1 1394.35
   177.1 1394.08   182.1 1394.37     187 1394.64   206.6 1399.11   216.5 1400.47
   255.8 1402.71   265.7 1403.45   275.5 1405.15   285.4 1408.67   295.1 1412.64
     344 1433.59   363.5 1442.18   383.1 1451.01   392.8 1455.56   402.6 1460.28
   431.9 1474.86   441.7 1479.43   451.5 1483.68   461.2 1487.59   510.1 1505.53
#Mann= 3 , 0 , 0
       0     .08       0   172.1    .045       0   182.1     .08       0
Bank Sta=172.1,182.1
XS Rating Curve= 0 ,0
Exp/Cntr=0.3,0.1

Type RM Length L Ch R = 1 ,36503.2 ,456.6,466,473.3
XS GIS Cut Line= 3
     1769142.696      145255.355     1769236.843      145556.628
     1769347.938      145695.967
#Sta/Elev= 30
     9.9 1431.93    19.7 1426.07    29.6 1420.39    49.3 1409.48    59.2 1404.66
      69 1401.49    78.9 1400.49    88.8 1400.09   118.4 1399.07     148 1398.56
   157.8 1397.98   167.7 1396.25   177.5 1393.63   187.4  1391.5   192.3 1391.37
   197.3 1391.24   202.3  1391.8   207.1 1392.33   226.9 1395.09   266.3  1397.9
     286  1399.5   315.6 1401.08     375 1403.09   384.9 1403.57   394.8 1404.29
   404.7 1405.26   434.4 1409.27   444.3  1410.4   464.1 1412.29   493.8 1414.41
#Mann= 3 , 0 , 0
       0      .1       0   192.3    .045       0   202.3      .1       0
Bank Sta=192.3,202.3
XS Rating Curve= 0 ,0
Exp/Cntr=0.3,0.1

Type RM Length L Ch R = 1 ,36037.1 ,381.7,394.7,407.7
XS GIS Cut Line= 3
     1768867.259      145220.931     1768835.888      145353.778
     1768804.517      145486.624
#Sta/Elev= 30
     9.7  1442.9    19.5 1436.61    29.2  1430.2      39 1423.82    48.8 1417.51
    58.5  1411.3    68.2 1405.55      78 1401.15    87.7 1398.67    97.5 1397.41
   107.3 1396.14     117 1394.06   126.8 1391.11   136.5 1388.74   141.2 1388.31
   146.2 1387.86   151.2 1388.01     156 1388.16   165.7 1389.21   175.5 1390.56
   185.3 1391.68     195 1392.78   204.7 1393.91   214.5 1395.29   224.2 1397.61
     234 1400.85   243.8 1404.52   253.5 1408.36   263.3 1412.29     273 1416.22
#Mann= 3 , 0 , 0
       0      .1       0   141.2    .045       0   151.2      .1       0
Bank Sta=141.2,151.2
XS Rating Curve= 0 ,0
Exp/Cntr=0.3,0.1

Type RM Length L Ch R = 1 ,35642.4 ,368.8,367.6,366.4
XS GIS Cut Line= 3
     1768632.922      145061.962     1768450.127      145214.292
     1768398.411      145269.432
#Sta/Elev= 18
     9.9 1413.88    19.8 1411.19    29.7  1408.7    49.6 1404.09    69.4 1400.46
    79.3  1398.8    99.1 1395.75     119 1393.12   168.5 1387.14   173.5 1386.96
   178.5 1386.77   183.5 1387.13   188.4 1387.48   198.3 1389.71   208.2  1392.5
   237.9 1400.14   256.8 1404.83   313.5 1417.78
#Mann= 3 , 0 , 0
       0      .1       0   173.5    .045       0   183.5      .1       0
Bank Sta=173.5,183.5
XS Rating Curve= 0 ,0
Exp/Cntr=0.3,0.1

Type RM Length L Ch R = 1 ,35274.9 ,489.2,481.5,473.8
XS GIS Cut Line= 2
     1768444.119      144758.254     1768218.164      144954.082
#Sta/Elev= 24
      10 1403.53    19.9 1399.18    29.9 1396.61    39.9 1395.33    59.8 1393.19
    89.7 1390.59   129.6 1387.24   149.5 1385.27   159.5  1384.7   169.4 1384.44
   174.4 1384.43   179.4 1384.42   184.4 1384.95   189.4 1385.49   199.3 1387.47
   219.3 1392.35   229.2 1394.88   239.2 1397.75   249.2  1401.1   259.1 1404.94
   269.1 1409.29   279.1 1414.05     289 1419.28     299    1425
#Mann= 3 , 0 , 0
       0      .1       0   174.4    .045       0   184.4      .1       0
Bank Sta=174.4,184.4
XS Rating Curve= 0 ,0
Exp/Cntr=0.3,0.1

Type RM Length L Ch R = 1 ,34793.4 ,436.1,427.7,418.9
XS GIS Cut Line= 2
     1768072.181      144430.029     1767916.837      144766.608
#Sta/Elev= 26
      10 1451.82      20 1443.49    40.1 1426.93    50.1 1418.06    60.1 1407.11
    70.1 1394.91    80.2  1386.2    85.2 1385.05    90.2  1383.9    95.2 1384.24
   120.2 1385.99   160.3 1388.22   170.3 1388.67   180.3 1388.74   190.4 1388.56
   200.4 1388.26   220.4 1387.25   230.4    1387   240.5 1387.06   260.5 1387.52
   290.5 1388.64   300.6 1389.27   310.6 1391.05   320.6 1394.42   330.6 1398.72
   370.7 1416.51
#Mann= 3 , 0 , 0
       0      .1       0    85.2    .045       0    95.2      .1       0
Bank Sta=85.2,95.2
XS Rating Curve= 0 ,0
Exp/Cntr=0.3,0.1

Type RM Length L Ch R = 1 ,34365.7 ,306.5,323.8,341.6
XS GIS Cut Line= 2
     1767612.112      144480.209     1767616.819      144743.823
#Sta/Elev= 29
     9.8 1406.34    19.5 1404.37    29.3 1402.19    39.1 1399.67    48.8 1396.52
    58.6 1392.56    68.4 1388.55    78.1 1385.68    87.9 1384.34    92.6 1384.34
    97.7 1383.88   102.6 1384.97   107.4 1385.58   117.2 1387.68   126.9 1389.97
   136.7 1392.03   146.5 1393.92   156.2 1395.84     166 1397.71   175.8 1399.56
   185.5 1401.51   195.3 1404.26   205.1 1408.44   214.8 1413.79   224.6  1419.5
   234.4 1425.24   244.1 1430.53   253.9 1434.98   263.7 1438.87
#Mann= 3 , 0 , 0
     9.8      .1       0    92.6    .045       0   102.6      .1       0
Bank Sta=92.6,102.6
XS Rating Curve= 0 ,0
Exp/Cntr=0.3,0.1

Type RM Length L Ch R = 1 ,34041.9 ,410.1,396.8,383.4
XS GIS Cut Line= 2
     1767469.454      144398.845     1767224.669       144605.97
#Sta/Elev= 25
      10 1391.06      20 1389.77    40.1 1387.55    50.1  1386.7    60.1  1386.3
   100.2 1385.77   120.2  1385.4   140.3 1384.87   150.3 1384.53   170.3 1383.62
   180.4 1382.72   190.4 1381.47   195.4 1381.35   200.4 1381.24   205.4 1382.81
   210.4 1384.38   230.5 1395.59   240.5 1401.41   250.5 1409.13   260.5  1418.3
   280.6 1437.07   290.6 1446.25   300.6 1455.02   310.6 1462.69   320.7 1469.18
#Mann= 3 , 0 , 0
       0      .1       0   195.4    .045       0   205.4      .1       0
Bank Sta=195.4,205.4
XS Rating Curve= 0 ,0
Exp/Cntr=0.3,0.1

Type RM Length L Ch R = 1 ,33645.1 ,696.2,691.9,687.3
XS GIS Cut Line= 2
     1767095.216      144071.681      1767015.19       144434.15
#Sta/Elev= 28
      10 1411.88    20.1 1408.42    30.1 1405.19    40.1 1402.18    60.2 1396.69
    70.2 1394.19    80.3 1391.91    90.3 1389.82   110.4 1385.94   120.4 1384.16
   130.4 1382.52   140.5 1381.16   150.5  1379.7   160.5 1378.13   170.6 1377.03
   175.6 1376.92   180.6 1376.81   185.6 1377.13   190.6 1377.44   200.6 1378.65
   260.8 1386.37     311  1393.2     321  1394.7   331.1  1397.2   341.1 1401.52
   351.1 1407.05   361.2 1412.99   371.2 1419.09
#Mann= 3 , 0 , 0
       0      .1       0   175.6    .045       0   185.6      .1       0
Bank Sta=175.6,185.6
XS Rating Curve= 0 ,0
Exp/Cntr=0.3,0.1

Type RM Length L Ch R = 1 ,32953.2 ,377.7,372.9,368.1
XS GIS Cut Line= 2
     1766389.107      144017.546     1766391.461      144356.479
#Sta/Elev= 28
      10 1395.92    19.9 1394.08    29.9 1392.39    39.9 1391.12    49.8 1390.35
    59.8 1389.69    69.8 1388.72    79.8 1387.19   119.6 1379.23   129.6 1377.11
   139.6 1374.83   149.5 1372.84   159.5 1371.53   169.5 1370.81   209.3 1368.58
   214.3 1368.56   219.3 1368.54   224.3 1369.22   229.3  1369.9   249.2 1374.49
   259.2 1376.54   269.2 1378.42   279.1 1380.56   289.1 1384.14   299.1 1390.16
     309 1398.04     319 1406.36   338.9 1422.54
#Mann= 3 , 0 , 0
       0      .1       0   214.3    .045       0   224.3      .1       0
Bank Sta=214.3,224.3
XS Rating Curve= 0 ,0
Exp/Cntr=0.3,0.1

Type RM Length L Ch R = 1 ,32580.3 ,272.3,251.1,230
XS GIS Cut Line= 3
      1765944.75      143947.267     1766065.289      144388.654
     1766107.655      144433.374
#Sta/Elev= 30
     9.9 1448.01    19.9 1444.33    39.8 1436.57    59.7 1428.38    69.6 1424.07
    79.6 1419.54    99.5 1409.91   129.3 1394.11   149.2 1383.92   159.1 1379.26
   169.1 1375.08     179 1372.18     189 1371.24   208.9 1370.66   228.8 1369.84
   268.6 1367.87   318.3 1365.18   333.2 1364.61   338.2 1364.49   343.2 1364.59
   348.1 1364.69   358.1 1365.73     378 1369.72   397.9 1372.65   417.8  1375.2
   427.7 1376.76   437.7 1379.12   457.5 1385.37   475.2 1392.12   519.2 1408.49
#Mann= 3 , 0 , 0
       0      .1       0   333.2    .045       0   343.2      .1       0
Bank Sta=333.2,343.2
XS Rating Curve= 0 ,0
Exp/Cntr=0.3,0.1

Type RM Length L Ch R = 1 ,32329.2 ,308,304.7,301.4
XS GIS Cut Line= 3
     1765369.481      144199.955     1765592.632      144374.265
     1766017.224      144485.932
#Sta/Elev= 30
    10.1 1418.39    50.6 1423.39    60.7 1424.02    70.8 1422.43    80.9 1417.35
   101.1 1404.84   111.2 1400.33   131.5 1394.35   192.1 1385.01   212.4 1382.92
   242.7 1382.96   262.9  1380.3   283.2 1374.09   313.1 1367.43     343 1357.52
     353 1355.78     363 1355.92     373 1357.69   402.9 1367.91   422.9 1369.79
   472.7 1370.11   552.6 1365.76  579.88 1365.15  584.67 1364.48   590.2  1365.2
   602.5 1365.89   612.4 1367.66   652.3 1377.32   692.3 1381.48   722.2 1387.28
#Mann= 3 , 0 , 0
    10.1      .1       0  579.88    .045       0   590.2      .1       0
#XS Ineff= 2 , 0
          455.03  1374.5
Permanent Ineff=
       F       F
Bank Sta=579.88,590.2
XS Rating Curve= 0 ,0
Exp/Cntr=0.3,0.1

Type RM Length L Ch R = 1 ,32024.5 ,602.4,608.3,614.2
XS GIS Cut Line= 2
     1765193.854      144673.073     1766024.285      144740.131
#Sta/Elev= 30
      10  1542.8    80.3 1518.31    90.3 1514.32   100.4  1509.3   110.4 1503.32
   140.5 1484.62   160.6 1472.54   170.6  1466.7   190.7 1455.34   210.8 1444.28
   281.1 1406.94   351.3 1369.41   361.4 1364.58   371.4 1361.08   381.4 1359.18
   391.5  1358.3   411.5 1357.19   421.6 1356.83   481.8 1355.69   582.2 1354.29
   677.6 1353.31   682.6 1353.27   687.6 1353.29   692.6  1353.3   702.6 1354.28
   712.7 1357.45   722.7 1362.29   732.8 1366.93   772.9 1383.12   833.1 1407.75
#Mann= 3 , 0 , 0
       0      .1       0   677.6    .045       0   687.6      .1       0
Bank Sta=677.6,687.6
XS Rating Curve= 0 ,0
Exp/Cntr=0.3,0.1

Type RM Length L Ch R = 1 ,31416.1 ,214.8,218.3,221.8
XS GIS Cut Line= 2
     1765595.912      145260.298     1765904.246      145375.629
#Sta/Elev= 21
      10 1375.48    59.9 1358.55    69.8  1355.5    79.8 1353.33    89.8 1351.96
   109.7 1349.45   119.7  1347.9   129.7 1346.63   134.7 1346.39   139.7 1346.15
   144.7 1346.29   149.6 1346.43   159.6 1347.58   169.6 1349.13   179.6 1350.55
   199.5  1353.2   239.4 1358.71   279.3 1363.87   289.3  1365.1   319.2 1368.47
   329.2 1369.85
#Mann= 3 , 0 , 0
       0      .1       0   134.7    .045       0   144.7      .1       0
Bank Sta=134.7,144.7
XS Rating Curve= 0 ,0
Exp/Cntr=0.3,0.1

Type RM Length L Ch R = 1 ,31197.8 ,309.3,313.1,316.9
XS GIS Cut Line= 3
     1765517.591      145432.228     1765746.549      145570.985
     1765786.561       145625.12
#Sta/Elev= 27
     9.9 1377.12    49.6 1360.51    59.5 1356.71    69.4 1354.23    79.3 1352.87
   109.1 1349.64     119 1348.48   128.9 1347.18   138.8 1346.29   143.7 1346.18
   148.7 1346.07   153.7 1346.33   158.7 1346.59   168.6 1348.06   178.5 1349.97
   188.4 1351.45   208.2 1354.22   228.1 1357.11     238 1358.71   247.9 1360.78
   257.8 1363.37   277.3 1368.68     287 1371.12   306.2 1375.55   315.8  1377.9
   325.4 1380.37     335 1383.32
#Mann= 3 , 0 , 0
       0      .1       0   143.7    .045       0   153.7      .1       0
Bank Sta=143.7,153.7
XS Rating Curve= 0 ,0
Exp/Cntr=0.3,0.1

Type RM Length L Ch R = 1 ,30884.7 ,655.6,655,654.3
XS GIS Cut Line= 2
     1765236.865      145531.496     1765598.266      145844.014
#Sta/Elev= 30
      10 1407.22    39.8 1393.82    49.8  1389.7    59.7 1387.16    69.7 1385.77
    99.5 1383.09   109.5 1381.98   119.4 1379.95   129.4 1377.05   189.1 1356.92
   199.1 1353.89     209 1351.71     219 1350.69   268.8 1347.37   288.7 1345.84
   293.6  1345.7   298.6 1345.54   303.6 1345.57   308.6  1345.6   318.5 1346.03
   338.4 1348.05   388.2  1352.5   398.2 1353.54   408.1 1354.75   418.1 1356.28
     428 1358.14     438  1360.5   447.9  1363.9   457.9 1367.62   477.8 1375.63
#Mann= 3 , 0 , 0
       0      .1       0   293.6    .045       0   303.6      .1       0
Bank Sta=293.6,303.6
XS Rating Curve= 0 ,0
Exp/Cntr=0.3,0.1

Type RM Length L Ch R = 1 ,30229.7 ,473.7,461.1,448.4
XS GIS Cut Line= 2
     1764870.974       145949.93     1765071.038      146109.982
#Sta/Elev= 28
     9.9 1370.79    19.7 1368.01    29.6 1365.25    39.4 1362.52    49.3 1359.82
    59.1 1357.13      69 1354.42    78.8 1351.74    88.7 1349.09    98.5  1346.1
   108.4 1343.38   113.2 1342.73   118.2 1342.05   123.2 1342.15   128.1 1342.25
     138 1345.47   147.8 1349.89   157.7 1352.22   167.5 1351.69   177.4 1351.93
   187.2 1354.72   197.1 1358.37   206.9  1362.2   216.8 1365.78   226.6 1369.64
   236.5 1373.16   246.4 1376.69   256.2 1380.23
#Mann= 3 , 0 , 0
       0      .1       0   113.2    .045       0   123.2      .1       0
Bank Sta=113.2,123.2
XS Rating Curve= 0 ,0
Exp/Cntr=0.3,0.1

Type RM Length L Ch R = 1 ,29768.7 ,597.4,608.8,620.2
XS GIS Cut Line= 4
     1764586.177      146286.509     1764720.337      146418.316
     1765002.781      146432.438      1765167.54      146477.158
#Sta/Elev= 30
     9.9 1471.81    39.6 1462.15    59.4 1455.13   128.7 1428.55   188.1 1407.49
   208.3 1394.87   218.4 1388.36   228.5 1381.45   248.7 1366.29   268.9 1350.46
     279 1344.19   284.1 1343.03   289.1 1341.91   294.1 1342.21   299.2 1342.52
   309.3 1344.83   319.4 1347.59   329.5 1348.96   349.7 1348.63   359.8 1348.74
   369.9 1349.69   440.6 1359.29   460.8 1362.54     491 1369.52   521.1 1377.45
   551.2 1385.96   591.4 1397.76   621.5 1406.07   631.5 1409.02   641.6 1412.47
#Mann= 3 , 0 , 0
     9.9      .1       0   284.1    .045       0   294.1      .1       0
#XS Ineff= 2 , 0
                          330.03          1352.4
Permanent Ineff=
       F       F
Bank Sta=284.1,294.1
XS Rating Curve= 0 ,0
Exp/Cntr=0.3,0.1

Type RM Length L Ch R = 1 ,29159.8 ,363.3,361.4,359.5
XS GIS Cut Line= 3
     1764449.663      146856.103     1764732.106       147051.46
     1764870.974      147079.704
#Sta/Elev= 30
    10.1 1368.42    40.4  1350.4    50.5 1344.89    60.6 1340.91    70.7 1339.34
    80.8 1338.79     101 1338.05   171.7 1334.73   176.8 1334.61   181.8 1334.49
   186.8 1334.63   191.9 1334.77     202 1335.97   222.2 1339.26   242.4 1341.26
   252.5 1342.56   262.6  1344.6   272.7 1346.98   282.8  1349.7   292.9 1352.69
     303 1355.94   323.2 1363.17   343.4 1371.05   362.3 1376.92   390.7 1385.17
   400.1 1388.43   409.6 1392.52   428.4 1402.02   437.9 1407.07   485.1 1433.08
#Mann= 3 , 0 , 0
       0      .1       0   176.8    .045       0   186.8      .1       0
Bank Sta=176.8,186.8
XS Rating Curve= 0 ,0
Exp/Cntr=0.3,0.1

Type RM Length L Ch R = 1 ,28798.4 ,435.4,435,434.6
XS GIS Cut Line= 2
     1764254.306       147159.73     1764503.798      147303.305
#Sta/Elev= 23
     9.9 1360.04    19.9 1353.43    29.8 1346.77    39.7 1340.74    49.6 1336.34
    59.6  1334.3    69.5  1333.7    89.3 1333.49    99.3 1332.92   109.2 1332.15
   119.1 1331.54     124 1331.46     129 1331.39     134 1331.62     139 1331.86
   148.9  1332.7   168.7 1334.64   198.5 1337.34   208.4  1338.4   218.4 1340.74
   228.3 1344.17   258.1 1355.48   287.9 1366.58
#Mann= 3 , 0 , 0
       0      .1       0     124    .045       0     134      .1       0
Bank Sta=124,134
XS Rating Curve= 0 ,0
Exp/Cntr=0.3,0.1

Type RM Length L Ch R = 1 ,28363.4 ,412.2,413.2,414.3
XS GIS Cut Line= 2
      1764021.29      147517.491     1764249.598      147639.883
#Sta/Elev= 28
      10 1352.35    19.9 1347.51    29.9 1342.64    39.9 1337.64    49.8 1332.72
    59.8 1329.58    69.7  1328.7    79.7 1328.37    89.7 1328.06    99.6 1327.78
   109.6 1327.49   119.6 1327.18   129.5 1326.85   139.5 1326.51   149.4  1326.1
   159.4 1325.65   164.4 1325.56   169.4 1325.48   174.4 1325.82   179.3 1326.15
   189.3 1327.88   199.3 1330.03   209.2 1332.01   219.2 1333.97   229.2 1336.38
   239.1 1339.44   249.1 1342.51     259 1345.43
#Mann= 3 , 0 , 0
       0      .1       0   164.4    .045       0   174.4      .1       0
Bank Sta=164.4,174.4
XS Rating Curve= 0 ,0
Exp/Cntr=0.3,0.1

Type RM Length L Ch R = 1 ,27950.2 ,495.9,493.3,490.8
XS GIS Cut Line= 2
     1763745.908      147776.398     1764009.521      147941.156
#Sta/Elev= 20
      10 1377.05    30.1 1360.51    40.1 1352.36    50.1 1344.33    60.2 1336.54
    70.2 1330.56    80.2 1327.03    90.3 1324.53   100.3 1322.22   110.3  1320.7
   115.3 1320.41   120.3 1320.12   125.3 1320.34   130.4 1320.57   140.4 1321.35
   180.5 1324.87   190.5 1325.82   250.7  1331.9   290.8 1336.19   310.9 1338.45
#Mann= 3 , 0 , 0
       0      .1       0   115.3    .045       0   125.3      .1       0
Bank Sta=115.3,125.3
XS Rating Curve= 0 ,0
Exp/Cntr=0.3,0.1

Type RM Length L Ch R = 1 ,27456.8 ,324.2,320.4,316.7
XS GIS Cut Line= 4
     1763503.452      148124.521     1763567.002       148244.56
     1763778.084      148341.532     1763853.352      148337.948
#Sta/Elev= 30
     9.7  1363.3    29.1  1355.4    38.8 1351.62    58.2 1344.69    77.6  1338.7
    87.3 1336.11      97 1333.68   106.7 1331.52   116.4 1329.53   126.1 1327.77
   135.8 1326.38   166.1 1323.14   186.3 1321.35   216.6 1318.84   236.8 1316.86
   241.9 1316.61   246.9 1316.36   251.9 1316.44     257 1316.53   267.1 1317.31
   277.2 1318.39   337.8 1323.94   347.9 1325.15     358  1327.1   368.1 1329.88
   377.5 1332.18   396.4 1336.46   405.8 1338.44     434 1343.72   443.5 1345.69
#Mann= 3 , 0 , 0
       0      .1       0   241.9    .045       0   251.9      .1       0
Bank Sta=241.9,251.9
XS Rating Curve= 0 ,0
Exp/Cntr=0.3,0.1

Type RM Length L Ch R = 1 ,27136.4 ,446.3,454,461.8
XS GIS Cut Line= 4
     1763312.828      148444.847     1763446.542      148565.547
     1763623.515      148609.606     1763656.467      148628.435
#Sta/Elev= 26
      10 1336.03      20 1330.82      30 1326.41      40 1323.79      50 1323.23
    70.1 1322.86   100.1 1322.65   130.1  1322.7   160.1 1322.55   170.1 1322.46
   180.1 1322.09   199.3 1321.02   208.9 1320.29   276.1 1314.31   285.7 1313.55
   290.3 1313.39   295.3 1313.22   300.3 1313.48   304.9 1313.73   314.5 1315.56
   324.1 1318.43   333.7 1321.42   343.3  1325.2   352.9 1329.82   362.5 1334.62
   400.5 1354.93
#Mann= 3 , 0 , 0
       0      .1       0   290.3    .045       0   300.3      .1       0
Bank Sta=290.3,300.3
XS Rating Curve= 0 ,0
Exp/Cntr=0.3,0.1

Type RM Length L Ch R = 1 ,26682.4 ,463.1,472.8,482.6
XS GIS Cut Line= 2
     1763041.524      148769.848     1763426.829      149053.002
#Sta/Elev= 30
      10 1343.74    19.9 1336.99    29.9 1331.46    39.8 1326.53    49.8 1322.49
    59.8 1320.11    69.7 1318.73    79.7 1318.23    89.7 1318.36   109.6  1319.8
   119.5 1320.04   129.5 1319.63   179.3  1316.2   239.1 1312.27   298.8 1307.47
   308.8 1306.82   313.8 1306.79   318.8 1306.76   323.8 1307.02   328.7 1307.28
   338.7 1308.91   378.5 1317.92   388.5 1320.11   408.4 1324.41   428.4 1328.47
   438.3 1330.19   448.3 1331.75   458.2 1333.13   468.2 1334.33   478.2 1335.29
#Mann= 3 , 0 , 0
       0      .1       0   313.8    .045       0   323.8      .1       0
Bank Sta=313.8,323.8
XS Rating Curve= 0 ,0
Exp/Cntr=0.3,0.1

Type RM Length L Ch R = 1 ,26209.6 ,747.2,739.7,732.2
XS GIS Cut Line= 2
     1762860.918      149085.052     1762995.079      149358.081
#Sta/Elev= 22
     9.8 1313.58    39.3 1313.07    68.7  1312.9    98.1 1312.88   107.9  1312.8
   127.6 1312.47   137.4 1312.19   147.2 1311.77     157 1311.21   176.6 1309.77
   186.5 1308.82   196.3 1307.61   206.1 1306.03   210.9 1305.41   215.9 1304.76
   220.9 1304.81   225.7 1304.87   235.5 1306.64   245.3 1309.81   255.1  1313.9
     265 1318.47   304.2  1337.2
#Mann= 3 , 0 , 0
       0      .1       0   210.9    .045       0   220.9      .1       0
Bank Sta=210.9,220.9
XS Rating Curve= 0 ,0
Exp/Cntr=0.3,0.1

Type RM Length L Ch R = 1 ,25469.9 ,634,629.4,624.7
XS GIS Cut Line= 2
     1762170.557      149388.127     1762489.034      149680.537
#Sta/Elev= 26
    10.1 1347.27    20.1 1341.16    40.2 1329.09    60.3 1317.27    70.4 1310.91
    80.4 1303.83    90.5 1298.19    95.5  1297.4   100.5 1296.62   105.5 1296.65
   110.6 1296.68     191 1299.29   271.5 1301.66   281.5 1302.01   291.6 1302.78
   301.6 1303.93   321.8 1306.72   351.9 1311.06     362 1312.43     372 1313.28
   382.1 1312.78   392.1 1313.24   402.2 1316.04   412.2 1320.31   422.3 1323.85
   432.4 1327.72
#Mann= 3 , 0 , 0
       0      .1       0    95.5    .045       0   105.5      .1       0
Bank Sta=95.5,105.5
XS Rating Curve= 0 ,0
Exp/Cntr=0.3,0.1

Type RM Length L Ch R = 1 ,24840.5 ,443.9,440.4,436.9
XS GIS Cut Line= 2
     1761771.157      149897.077     1762140.687      150101.849
#Sta/Elev= 26
    10.1  1327.2    40.2 1318.56    50.3 1315.83    80.5  1308.1   100.6 1303.14
   130.8 1295.92   140.8  1293.1   150.9 1290.97   155.9 1290.54   160.9 1290.11
   165.9 1290.14     171 1290.17   201.2 1291.36   231.4 1292.37   261.5 1293.08
   271.6 1293.62   281.6 1294.81   301.8 1297.98   311.8 1300.56   321.9 1304.91
   331.9 1310.58     342 1316.72   352.1 1323.13   392.3 1350.11   412.4 1363.43
   422.5 1369.96
#Mann= 3 , 0 , 0
       0      .1       0   155.9    .045       0   165.9      .1       0
Bank Sta=155.9,165.9
XS Rating Curve= 0 ,0
Exp/Cntr=0.3,0.1

Type RM Length L Ch R = 1 ,24400.1 ,524,521.3,518.6
XS GIS Cut Line= 2
     1761540.852      150288.889     1761888.075      150421.057
#Sta/Elev= 30
      10  1337.3    20.1 1329.24    30.1  1321.9    40.2 1315.24    50.2 1309.35
    60.2 1304.31    70.3 1300.11    80.3 1296.67    90.4 1293.82   100.4  1291.4
   110.5 1289.47   120.5  1288.1   140.6 1285.57   145.6 1285.26   150.6 1284.94
   155.6 1284.95   160.7 1284.97   170.7 1285.74   200.8 1290.36   210.9 1291.64
   220.9 1292.61   230.9 1293.22     241  1293.5   271.1 1293.69   291.2 1294.27
   301.2 1296.14   311.3 1299.34   351.4 1313.27   361.5 1317.18   371.5 1321.53
#Mann= 3 , 0 , 0
       0      .1       0   145.6    .045       0   155.6      .1       0
Bank Sta=145.6,155.6
XS Rating Curve= 0 ,0
Exp/Cntr=0.3,0.1

Type RM Length L Ch R = 1 ,23878.9 ,239.4,242.4,245.3
XS GIS Cut Line= 2
      1761396.92      150782.067     1761806.463        150866.8
#Sta/Elev= 30
      10 1344.47    39.8 1325.56    59.7  1313.3    79.7 1301.42    89.6 1295.34
    99.6 1288.73   109.5 1282.63   119.5 1279.42   124.4 1279.38   129.4 1279.34
   134.4 1280.05   139.4 1280.76   169.3 1286.66   179.2 1288.43   189.2 1289.74
   199.2 1290.64   219.1 1292.08   248.9 1293.77   258.9 1294.17   278.8 1294.58
   298.7 1294.54   308.7 1294.25   328.6 1292.91   338.6 1293.69   348.5  1297.6
   358.5 1304.11   378.4 1318.69   398.3 1333.68   408.3 1341.35   418.2 1349.33
#Mann= 3 , 0 , 0
       0      .1       0   124.4    .045       0   134.4      .1       0
Bank Sta=124.4,134.4
XS Rating Curve= 0 ,0
Exp/Cntr=0.3,0.1

Type RM Length L Ch R = 1 ,23636.5 ,370.8,381.9,393
XS GIS Cut Line= 2
     1761323.955      150989.192     1761688.778      151118.645
#Sta/Elev= 30
     9.9 1348.66    19.9 1340.47    29.8 1331.67    49.6 1313.69    59.6 1305.39
    69.5 1298.35    79.4 1292.69    99.3 1282.29   109.2 1278.65   114.1 1278.14
   119.1 1277.62   124.1 1278.08     129 1278.54   148.9 1282.06   158.8 1283.33
   178.7 1284.47   188.6 1286.16   198.5    1288   208.4  1289.3   238.2 1292.16
   248.1 1293.55   258.1 1295.72     268 1298.45   287.9 1304.15   307.7 1310.25
   317.6 1312.34   327.6 1313.53   347.4 1315.52   377.2 1319.38   387.1 1320.54
#Mann= 3 , 0 , 0
       0      .1       0   114.1    .045       0   124.1      .1       0
Bank Sta=114.1,124.1
XS Rating Curve= 0 ,0
Exp/Cntr=0.3,0.1

Type RM Length L Ch R = 1 ,23254.6 ,396.5,396.7,396.9
XS GIS Cut Line= 2
     1761201.563      151252.806     1761401.627       151497.59
#Sta/Elev= 29
     9.9 1289.92    19.8 1289.39    29.6 1289.21    88.9  1288.8    98.8 1288.49
   108.7 1287.08   118.6 1283.97   128.4  1280.1   138.3 1276.78   143.2 1276.29
   148.2 1275.79   153.2 1275.97   158.1 1276.15   167.9 1277.39   177.8 1278.78
   187.7 1280.43   197.6 1282.77   207.5 1285.81   217.3 1289.39   227.2 1294.23
   237.1 1299.59     247 1305.43   256.9 1311.08   266.7 1316.38   276.6 1321.61
   286.5 1327.47   296.4 1333.81   306.3 1339.97   316.1 1345.89
#Mann= 3 , 0 , 0
       0      .1       0   143.2    .045       0   153.2      .1       0
Bank Sta=143.2,153.2
XS Rating Curve= 0 ,0
Exp/Cntr=0.3,0.1

Type RM Length L Ch R = 1 ,22857.9 ,431.7,430.2,428.7
XS GIS Cut Line= 3
     1760911.021      151513.828     1760995.833      151620.782
     1761080.645      151727.736
#Sta/Elev= 30
     9.8 1285.98    19.5 1285.76    29.2 1285.59      39 1285.44    48.7  1285.3
    58.5 1285.14    68.2 1284.94      78 1284.68    87.7 1284.44    97.5 1283.63
   107.2 1281.85     117 1279.19   126.7 1276.27   131.5 1275.31   136.5 1274.31
   141.5 1274.53   146.2 1274.73     156 1277.89   165.7 1283.79   175.5 1289.97
   185.2  1295.6     195 1301.14   204.7 1306.62   214.5 1312.13   224.2 1317.85
     234 1324.34   243.7 1332.29   253.5 1341.75   263.2 1351.69     273 1361.11
#Mann= 3 , 0 , 0
       0      .1       0   131.5    .045       0   141.5      .1       0
Bank Sta=131.5,141.5
XS Rating Curve= 0 ,0
Exp/Cntr=0.3,0.1

Type RM Length L Ch R = 1 ,22427.7 ,98.4,97.2,95.9
XS GIS Cut Line= 2
      1760575.48      151787.095     1760820.264      152064.831
#Sta/Elev= 30
      10 1289.77      20 1285.01      30 1282.37      40 1281.21      70 1278.79
      80  1277.9    90.1 1276.78   110.1 1273.99   120.1 1272.48   140.1 1268.96
   145.1 1268.53   150.1 1268.11   155.1 1268.25   160.1  1268.4   170.1 1269.82
   180.1 1271.39   190.1 1272.73   200.1 1273.93   220.1 1276.62   250.1 1280.23
   260.1  1282.2   270.2 1284.67   300.2 1292.74   310.2  1295.6   320.2  1298.6
   330.2 1301.73   340.2 1305.17   350.2 1308.91   360.2 1312.97   370.2 1317.61
#Mann= 3 , 0 , 0
       0      .1       0   145.1    .045       0   155.1      .1       0
Bank Sta=145.1,155.1
XS Rating Curve= 0 ,0
Exp/Cntr=0.3,0.1

Type RM Length L Ch R = 1 ,22330.5 ,390.8,405.2,419.3
XS GIS Cut Line= 3
     1760493.812      151853.985      1760695.04       152048.99
     1760768.568      152121.079
#Sta/Elev= 30
      10 1298.05      20 1291.46      30 1285.53      40 1281.45      50 1279.08
    80.1  1274.2    90.1 1272.36   100.1 1270.11   110.1 1268.07   115.1  1267.4
   120.1 1266.72   125.1 1266.89   130.1 1267.05   140.1 1268.66   160.1 1273.14
   170.1 1274.74   180.1 1275.92   190.1 1276.71   200.2 1277.13   210.2  1277.3
   230.2 1277.24   240.2 1277.51   250.2 1278.49   260.2 1280.82   280.2  1286.4
   308.3 1293.95   336.4 1301.23   364.5 1308.66   373.8 1311.22   383.2    1314
#Mann= 3 , 0 , 0
       0      .1       0   115.1    .045       0   125.1      .1       0
Bank Sta=115.1,125.1
XS Rating Curve= 0 ,0
Exp/Cntr=0.3,0.1

Type RM Length L Ch R = 1 ,21925.3 ,430.2,428.4,426.7
XS GIS Cut Line= 3
     1760264.792      152008.342     1760290.683      152069.538
     1760342.464       152363.75
#Sta/Elev= 29
     9.5 1306.23      19 1301.12    28.5 1296.17      38 1291.77    47.5 1287.85
      57 1284.17    66.4 1280.88    76.4 1278.47    86.4 1277.23    96.3 1276.45
   116.2 1275.28   146.1 1273.93   156.1 1273.36     166 1272.56     176 1270.78
   195.9 1264.52   200.9 1263.98   205.9 1263.45   210.9 1264.37   215.8 1265.27
   225.8 1268.95   235.7  1271.8   245.7 1273.16   305.4 1277.68   325.4 1278.97
   335.3 1279.79   345.3 1282.14   355.2 1286.74   365.2 1292.45
#Mann= 3 , 0 , 0
       0      .1       0   200.9    .045       0   210.9      .1       0
Bank Sta=200.9,210.9
XS Rating Curve= 0 ,0
Exp/Cntr=0.3,0.1

Type RM Length L Ch R = 1 ,21496.9 ,442.3,429.2,416.2
XS GIS Cut Line= 3
      1759881.14      152100.136     1759956.458      152403.763
     1759998.825      152436.714
#Sta/Elev= 29
    10.1 1276.07    40.4 1274.53   100.9  1271.8   121.1 1270.73   131.2 1270.07
   141.3 1268.91   151.4 1266.94   161.5 1264.14   171.6 1261.09   176.6 1260.14
   181.6 1259.18   186.6  1259.2   191.7 1259.23   201.8 1261.05     222 1266.39
   232.1  1269.7   242.2 1273.88   252.3 1278.93   262.4 1285.06   272.5 1293.03
   282.6 1302.12   292.6 1312.03   302.7 1322.57   312.8 1334.25   321.8 1344.01
   330.7 1351.51   339.7 1356.95   348.6 1361.15   366.5  1369.2
#Mann= 3 , 0 , 0
       0      .1       0   176.6    .045       0   186.6      .1       0
Bank Sta=176.6,186.6
XS Rating Curve= 0 ,0
Exp/Cntr=0.3,0.1

Type RM Length L Ch R = 1 ,21067.7 ,313.5,309.7,305.9
XS GIS Cut Line= 3
     1759412.755      152215.467     1759629.295      152399.055
     1759746.979      152462.605
#Sta/Elev= 30
     9.8 1272.82    29.4  1271.7    48.9 1270.43    58.7 1269.66    78.3 1267.77
    88.1 1266.22    97.9 1262.54   107.7 1258.55   112.5  1257.4   117.5 1256.21
   122.5 1256.36   127.3  1256.5   137.1 1258.38   146.8  1260.8   156.6  1262.7
   166.4 1264.24   176.2 1265.27     186 1265.86   244.7 1268.16   293.4 1269.93
     303 1270.61   312.6  1272.5   322.1 1277.35   331.7 1284.43   350.8  1300.9
   360.3 1308.71   369.9 1315.86   379.4 1322.46   408.1 1341.34   417.6  1347.8
#Mann= 3 , 0 , 0
       0      .1       0   112.5    .045       0   122.5      .1       0
Bank Sta=112.5,122.5
XS Rating Curve= 0 ,0
Exp/Cntr=0.3,0.1

Type RM Length L Ch R = 1 ,20758   ,86.2,83.6,81
XS GIS Cut Line= 2
     1759197.751       152472.46     1759516.293      152645.414
#Sta/Elev= 24
    10.1  1307.8    30.2 1301.44    50.3 1295.62    60.4 1292.05    70.5 1287.59
    80.5 1282.62   110.8 1266.96   120.8 1261.46   130.9  1256.3     136 1254.84
     141 1253.41     146 1253.54     151 1253.67   161.1 1256.85   171.2  1260.8
   181.2 1262.19   241.6 1262.25   302.1 1262.15   312.1 1262.27   322.2 1263.23
   332.3 1266.38   342.3 1271.57   352.4 1277.28   362.5 1283.18
#Mann= 3 , 0 , 0
       0      .1       0     136    .045       0     146      .1       0
Bank Sta=136,146
XS Rating Curve= 0 ,0
Exp/Cntr=0.3,0.1

Type RM Length L Ch R = 1 ,20674.4 ,262.7,256.4,250.1
XS GIS Cut Line= 3
     1759128.218      152555.914     1759337.436      152636.779
     1759509.256      152728.573
#Sta/Elev= 29
     9.8 1302.89    19.5 1301.55      39 1299.54    48.8 1298.43    58.5 1297.11
    68.3 1295.58      78 1293.83    87.8 1291.63    97.5 1288.39   107.3 1283.85
     117 1278.51   136.5  1267.5     156 1255.75   160.8 1253.95   165.8 1252.06
   170.8 1252.09   175.5 1252.12   185.3  1255.3     195 1258.99   204.8 1260.69
   214.5 1260.95   331.4 1261.96   341.2 1262.24   350.9  1263.5   360.7 1266.94
   389.9 1279.65   399.6 1284.13   409.4 1288.98   419.1 1294.28
#Mann= 3 , 0 , 0
       0      .1       0   160.8    .045       0   170.8      .1       0
Bank Sta=160.8,170.8
XS Rating Curve= 0 ,0
Exp/Cntr=0.3,0.1

Type RM Length L Ch R = 1 ,20418   ,316.3,315.6,314.9
XS GIS Cut Line= 2
     1759149.141      152862.733      1759403.34      152876.855
#Sta/Elev= 28
     9.8 1288.61    19.6 1284.96    29.4 1281.62    39.2 1277.91      49 1273.02
    58.8 1266.69    68.5 1259.37    78.3 1252.51    88.1 1248.71    92.9 1248.65
    97.9 1248.59   102.9 1249.33   107.7 1250.05   117.5 1251.46   127.3 1252.61
   137.1  1253.8   146.9 1255.11   156.7 1256.28   166.5 1257.07   176.3 1257.72
     186 1258.27   195.8 1258.77   205.6  1259.3   215.4 1259.94   225.2 1260.62
     235 1261.57   244.8 1263.88   254.6 1267.96
#Mann= 3 , 0 , 0
       0      .1       0    92.9    .045       0   102.9      .1       0
Bank Sta=92.9,102.9
XS Rating Curve= 0 ,0
Exp/Cntr=0.3,0.1

Type RM Length L Ch R = 1 ,20102.4 ,234,233.7,233.4
XS GIS Cut Line= 3
      1759180.18       153180.21     1759316.637      153183.664
     1759453.093      153187.119
#Sta/Elev= 30
     9.8 1258.32    19.5 1257.63    29.3 1256.91      39 1255.83    48.8 1253.77
    58.5 1250.57    68.3 1247.09      78 1244.82    82.8  1244.6    87.8 1244.37
    92.8 1244.85    97.5 1245.29   107.2 1247.05     117 1248.92   126.7 1250.62
   136.5  1252.3   146.3 1253.97     156 1255.62   165.8  1257.2   175.5 1258.67
   185.3 1259.38     195 1258.76   204.8 1257.32   214.5  1256.3   224.3 1256.56
     234 1257.69   243.8 1259.88   253.5 1263.83   263.3 1269.77     273 1277.31
#Mann= 3 , 0 , 0
       0      .1       0    82.8    .045       0    92.8      .1       0
Bank Sta=82.8,92.8
XS Rating Curve= 0 ,0
Exp/Cntr=0.3,0.1

Type RM Length L Ch R = 1 ,19868.7 ,472,470.8,469.6
XS GIS Cut Line= 3
     1759146.787      153413.498     1759393.925      153415.852
     1759631.648      153420.559
#Sta/Elev= 30
     9.9  1254.4    79.1 1252.03      89 1251.46    98.9 1250.23   118.6 1246.46
   128.5 1244.29   138.4 1242.54   143.3 1242.23   148.3 1241.91   153.3 1242.23
   158.2 1242.54   168.1 1244.24   177.9 1246.33   197.7 1250.11   217.5 1253.25
     267 1258.21   296.7 1261.47   306.6 1262.81   316.5 1264.65   326.4 1267.05
   385.8 1283.07   405.7 1288.79   415.6 1291.96   425.5  1295.9   435.4 1301.31
   445.3 1307.84   455.2 1314.05   465.1 1319.27     475  1323.7   484.9 1327.71
#Mann= 3 , 0 , 0
       0      .1       0   143.3    .045       0   153.3      .1       0
Bank Sta=143.3,153.3
XS Rating Curve= 0 ,0
Exp/Cntr=0.3,0.1

Type RM Length L Ch R = 1 ,19397.9 ,351.3,352.3,353.2
XS GIS Cut Line= 4
     1759095.573      153868.236      1759152.86      153870.878
     1759446.318      153857.437     1759620.447      153830.577
#Sta/Elev= 30
     9.6 1310.42    28.7 1299.48    38.2 1293.41    57.3 1280.53    76.9 1266.19
    86.7 1259.95    96.5 1255.01   106.3 1251.14   125.9 1244.77   135.7 1241.93
   145.5 1240.24   150.3 1240.09   155.3 1239.94   160.3 1240.32   165.1 1240.69
   174.9 1242.09   194.4 1245.21     214 1248.75   223.8    1250   282.6 1255.67
   321.7 1258.84   409.8 1265.13   439.2 1267.51     449 1268.17   478.4 1269.18
   488.1 1269.81   497.9 1271.44   507.7 1275.09   517.5 1280.84   527.3 1287.33
#Mann= 3 , 0 , 0
       0      .1       0   150.3    .045       0   160.3      .1       0
Bank Sta=150.3,160.3
XS Rating Curve= 0 ,0
Exp/Cntr=0.3,0.1

Type RM Length L Ch R = 1 ,19045.6 ,351,349.3,347.6
XS GIS Cut Line= 2
     1759081.175       154215.86     1759413.436      154215.448
#Sta/Elev= 29
    10.1 1288.46    30.2 1277.17    40.3 1271.69    50.3 1266.44    60.4 1261.38
    70.5  1256.7    80.5 1253.21    90.6 1251.05   110.8 1248.01   130.9 1244.56
     141 1242.67     151 1240.52   161.1 1238.57   166.2 1238.12   171.2 1237.69
   176.2 1237.96   181.2 1238.24   191.3 1239.98   201.4  1242.1   211.4  1243.9
   221.5 1245.24   231.6 1246.37   241.6 1247.35   251.7 1248.19   261.8 1248.89
   271.8 1249.42   281.9 1249.77     292 1249.99   332.3 1250.61
#Mann= 3 , 0 , 0
       0      .1       0   166.2    .045       0   176.2      .1       0
Bank Sta=166.2,176.2
XS Rating Curve= 0 ,0
Exp/Cntr=0.3,0.1

Type RM Length L Ch R = 1 ,18696.3 ,259.3,262.3,265.4
XS GIS Cut Line= 2
     1759085.591      154578.577     1759450.414      154547.979
#Sta/Elev= 30
     9.9 1250.67    19.8 1248.31    29.7 1246.36    39.6 1244.78    49.5 1243.83
    59.4 1243.35    69.3 1243.04    89.1 1242.84   118.7 1242.07   138.5 1241.88
   148.4 1241.59   158.3 1241.06   168.2 1240.24   178.1 1239.14     188 1237.92
   207.8 1235.02   217.7  1233.8   222.6 1233.61   227.6 1233.41   232.6 1233.82
   237.5 1234.22   247.4 1236.19   257.3 1238.56   277.1 1242.96   286.9 1245.68
   296.8 1249.55   306.7 1254.48   316.6  1259.7   326.5 1264.77   366.1 1284.24
#Mann= 3 , 0 , 0
       0      .1       0   222.6    .045       0   232.6      .1       0
Bank Sta=222.6,232.6
XS Rating Curve= 0 ,0
Exp/Cntr=0.3,0.1

Type RM Length L Ch R = 1 ,18434   ,562.1,563,563.7
XS GIS Cut Line= 2
     1759097.359      154811.593     1759483.365      154823.361
#Sta/Elev= 30
     9.9 1246.57    19.8 1244.11    29.7 1243.15    49.5 1242.42    69.3 1241.47
    79.2 1241.28      99  1241.7   108.9 1241.49   118.8 1240.06   128.7 1236.46
   138.6 1232.17   148.5 1229.85   153.4 1229.75   158.4 1229.64   163.4 1229.99
   168.3 1230.34   178.2 1231.35   227.8    1236   247.6 1238.04   267.4 1240.26
   277.3 1241.46   287.2  1242.8   297.1  1244.4     307 1246.25   316.9 1248.52
   326.8 1251.88   336.7 1256.51   346.6  1261.7   356.5 1267.05   386.2 1283.44
#Mann= 3 , 0 , 0
       0      .1       0   153.4    .045       0   163.4      .1       0
Bank Sta=153.4,163.4
XS Rating Curve= 0 ,0
Exp/Cntr=0.3,0.1

Type RM Length L Ch R = 1 ,17871   ,328.9,330,331
XS GIS Cut Line= 2
     1759108.198      155302.365     1759470.667      155342.377
#Sta/Elev= 25
     9.9 1242.52    19.7 1235.16    29.6 1232.91    88.7 1230.42   108.4 1229.92
   118.3 1229.88   167.6 1230.67   177.4 1230.65   187.3 1230.46   197.1 1230.12
   216.8 1229.08   236.5 1227.77   246.4 1227.02   256.3 1226.15   266.1 1225.13
     276 1224.21   280.8 1224.13   285.8 1224.05   290.8 1225.05   295.7 1226.04
   305.5 1230.95   315.4  1237.1   325.2 1242.32   335.1 1246.15   364.7 1255.77
#Mann= 3 , 0 , 0
       0      .1       0   280.8    .045       0   290.8      .1       0
Bank Sta=280.8,290.8
XS Rating Curve= 0 ,0
Exp/Cntr=0.3,0.1

Type RM Length L Ch R = 1 ,17541.1 ,416.3,424.6,433
XS GIS Cut Line= 2
     1758984.295      155599.863      1759430.91      155673.205
#Sta/Elev= 29
    10.1 1273.59    30.2 1260.31    50.3 1246.87    60.3 1240.31    70.4 1234.31
    80.5 1230.44    90.5 1229.22   191.1 1227.26   241.4 1226.38   251.4 1226.17
   261.5 1225.82   271.6 1225.28   291.7 1223.98   311.8 1222.48   321.8 1221.58
   326.9 1221.26   331.9 1220.95   336.9 1221.16     342 1221.38     352 1223.65
   362.1 1227.48   372.1  1231.7   382.2  1236.2   392.3  1241.5   402.3 1247.47
   422.4 1259.93   432.5 1265.75   442.5  1271.1   452.6 1276.04
#Mann= 3 , 0 , 0
       0      .1       0   326.9    .045       0   336.9      .1       0
Bank Sta=326.9,336.9
XS Rating Curve= 0 ,0
Exp/Cntr=0.3,0.1

Type RM Length L Ch R = 1 ,17116.4 ,331.4,336.5,341.5
XS GIS Cut Line= 2
     1758902.781      155867.137     1759229.785      156080.644
#Sta/Elev= 30
      10 1244.19      20 1238.05      30 1232.77    40.1  1229.7    50.1 1228.57
    70.1 1227.77   130.2 1225.67   180.2 1223.48   190.3 1223.25   200.3 1223.28
   210.3 1223.71   220.3 1224.01   230.3 1224.19   240.3 1223.79   250.3 1222.89
   260.4 1221.26   270.4 1218.96   280.4 1216.46   285.4 1215.68   290.4 1214.91
   295.4 1215.05   300.4 1215.19   310.4 1218.44   320.4 1223.85   330.5 1229.76
   340.5 1236.03   350.5 1242.98   360.5 1250.86   380.5 1268.28   390.5  1276.6
#Mann= 3 , 0 , 0
       0      .1       0   285.4    .045       0   295.4      .1       0
Bank Sta=285.4,295.4
XS Rating Curve= 0 ,0
Exp/Cntr=0.3,0.1

Type RM Length L Ch R = 1 ,16780   ,92.7,91.9,91
XS GIS Cut Line= 3
     1758730.183      156075.527     1758974.443      156331.087
       1759059.7      156317.958
#Sta/Elev= 30
    10.1 1241.86    30.3 1230.11    40.4 1225.87    50.5 1224.41    60.6 1224.11
     101 1223.75   161.6 1223.44     202 1222.77   212.1 1222.11   222.2 1220.72
   242.4 1215.62   252.5 1213.28   262.6 1211.52   267.7 1211.23   272.7 1210.95
   277.7 1211.21   282.8 1211.48   292.9 1213.36     303 1216.26   313.1 1218.87
   323.2 1221.03   333.3 1222.79   343.4    1224   372.7 1225.83   382.3 1227.55
   391.9 1232.39   401.4 1239.41     411 1246.18   420.6 1251.96   439.8 1262.38
#Mann= 3 , 0 , 0
       0      .1       0   267.7    .045       0   277.7      .1       0
Bank Sta=267.7,277.7
XS Rating Curve= 0 ,0
Exp/Cntr=0.3,0.1

Type RM Length L Ch R = 1 ,16688.1 ,198.1,200.2,202.2
XS GIS Cut Line= 2
     1758666.847      156144.997     1758943.793      156420.848
#Sta/Elev= 24
      10  1246.1      20 1239.04    30.1 1232.08    40.1 1226.02    50.1 1222.34
    60.1  1221.1    90.2 1220.53   120.3 1220.11   200.5  1219.3   210.5  1219.1
   220.5 1218.66   230.5 1217.84   270.6 1213.55   290.7 1211.22   300.7 1210.31
  305.46 1210.25   310.7 1210.77   315.7  1210.7   320.7 1211.16   330.8  1213.4
   350.8 1219.62   370.8 1225.46   380.9 1228.96   390.9 1233.32
#Mann= 3 , 0 , 0
      10      .1       0   300.7    .045       0   315.7      .1       0
#XS Ineff= 2 , 0
          196.46 1226.01
Permanent Ineff=
       F       F
Bank Sta=300.7,315.7
XS Rating Curve= 0 ,0
Exp/Cntr=0.3,0.1

Type RM Length L Ch R = 1 ,16488   ,295.7,302.5,309.3
XS GIS Cut Line= 2
       1758530.1       156240.95       1758799.3      156568.625
#Sta/Elev= 30
    10.1 1258.38    20.2 1251.39    30.3 1245.02    40.4 1239.23    60.6 1228.26
    70.7 1222.94    80.8 1219.44    90.9 1218.17   111.1 1217.82   181.7 1217.07
   222.1 1216.44   232.2 1216.37   242.3  1216.5   262.5 1217.02   272.6 1217.18
   282.7  1217.1   292.8 1216.64   302.9 1215.75     313 1214.24   323.1 1212.03
   328.2 1211.15  333.06 1210.13   338.2 1210.28   343.3 1210.28   353.4 1213.12
   363.5 1218.18   373.6 1223.77   383.7 1228.39   403.9 1236.73   424.1 1245.47
#Mann= 3 , 0 , 0
    10.1      .1       0   328.2    .045       0   338.2      .1       0
#XS Ineff= 2 , 0
          125.84 1227.34
Permanent Ineff=
       F       F
Bank Sta=328.2,338.2
XS Rating Curve= 0 ,0
Exp/Cntr=0.3,0.1

Type RM Length L Ch R = 1 ,16185.5 ,296.9,305.6,314.4
XS GIS Cut Line= 2
     1758392.183      156393.279     1758491.255      156663.555
#Sta/Elev= 23
     9.9 1230.81    19.9 1225.68    29.8  1220.9    39.7 1217.56    49.6 1216.46
    99.3 1214.33   109.2 1213.61     129 1211.87     139 1211.28   158.8 1210.35
   168.7 1210.15   188.6  1210.2   198.5 1210.04   208.5 1209.61   213.4 1209.55
   218.4 1209.48   223.4 1210.26   228.3 1211.02   238.2 1214.88   258.1 1224.74
     268 1229.82   277.9 1235.38   287.9 1241.14
#Mann= 3 , 0 , 0
       0      .1       0   213.4    .045       0   223.4      .1       0
Bank Sta=213.4,223.4
XS Rating Curve= 0 ,0
Exp/Cntr=0.3,0.1

Type RM Length L Ch R = 1 ,15879.9 ,302.7,312.5,322.4
XS GIS Cut Line= 2
     1758187.358      156444.803     1758162.716      156744.982
#Sta/Elev= 23
      10 1216.19    20.1 1214.75    30.1 1214.37    50.2 1214.03    80.3 1212.92
   100.4  1212.3   120.5 1211.41   140.6 1210.25   150.6 1209.57   170.7 1208.07
   190.8 1206.17   195.8 1206.02   200.8 1205.87   205.8 1206.68   210.8 1207.49
   220.9 1211.52     241 1222.25     251 1227.44     261 1232.56   271.1 1237.44
   281.1 1241.97   291.1 1246.08   301.2  1249.2
#Mann= 3 , 0 , 0
       0      .1       0   195.8    .045       0   205.8      .1       0
Bank Sta=195.8,205.8
XS Rating Curve= 0 ,0
Exp/Cntr=0.3,0.1

Type RM Length L Ch R = 1 ,15567.3 ,293.1,290.8,288.6
XS GIS Cut Line= 3
     1757981.605      156371.515     1757906.811      156485.702
     1757832.075      156599.923
#Sta/Elev= 30
     9.8 1212.98    19.5 1212.53    29.3 1211.88      39 1210.72    48.8 1209.04
    58.5 1207.21    68.3 1205.38      78 1203.62    87.8 1201.91    97.5 1200.13
   107.3 1198.37     112  1197.8     117 1197.19     122  1197.2   126.8 1197.21
   136.5 1198.86   146.3 1201.46     156 1204.04   165.8 1206.42   175.5 1209.04
   185.3 1211.91     195 1214.96   204.8  1218.1   214.5 1221.29   224.3  1224.5
     234 1227.76   243.8 1231.28   253.5 1235.35   263.3 1239.97     273 1244.84
#Mann= 3 , 0 , 0
       0      .1       0     112    .045       0     122      .1       0
Bank Sta=112,122
XS Rating Curve= 0 ,0
Exp/Cntr=0.3,0.1
